--- Buzzard Branch.prj (project) ---

Proj Title=Buzzard Branch
Current Plan=p01
Default Exp/Contr=0,0
English Units
Geom File=g01
Flow File=f01
Plan File=p01
BEGIN DESCRIPTION:
END DESCRIPTION:
DSS Export Rating Curves= 0
DSS Export Rating Curve Sorted= 0
DSS Export Volume Flow Curves= 0
DXF OffsetX= 0
DXF OffsetY= 0
DXF ScaleX= 0
DXF ScaleY= 0

--- Buzzard Branch.p01 (plan) ---

Plan Title=Floodplain
Program Version=4.00
Geom File=g01
Flow File=f01
K Sum by GR=0
Std Step Tol=0.01
Critical Tol=0.01
Num of Std Step Trials=20
Max Error Tol=0.3
Flow Tol Ratio=0.001
Split Flow NTrial=30
Split Flow Tol=0.02
Split Flow Ratio=0.02
Log Output Level=0
Friction Slope Method=1
Unsteady Friction Slope Method=2
Unsteady Bridges Friction Slope Method=1
Global Log Level=0
CheckData=False
Run HTab=0
Run UNet=0
Run PostProcess=0
UNET Theta=0
UNET Theta Warmup=0
UNET ZTol=0
UNET ZSATol=0
UNET MxIter=0
UNET MaxInSteps=0
UNET DtIC=0
UNET DtMin=0
UNET MaxCRTS=0
UNET WFStab=0
UNET SFStab=0
UNET WFX=0
UNET SFX=0
UNET DSS MLevel=0
UNET DZMax Abort=0
UNET Convert EG Bridges=0
UNET Use Existing IB Tables=0
UNET Froude Limit=0
UNET Froude Power=0
Write IC File=0
Echo Input=False
Echo Output=False
Write Detailed=0

--- Buzzard Branch.f01 (steady flow) ---

Flow Title=NFF Regression Equation
Program Version=4.00
Number of Profiles=1
Profile Names=P100yr
River Rch & RM=Buzzard Branch,Main      ,19045.3
601.1765
River Rch & RM=Buzzard Branch,Main      ,17132.9
652.4519
River Rch & RM=Buzzard Branch,Main      ,16845.2
832.9369
River Rch & RM=Buzzard Branch,Main      ,14416.2
922.0791
River Rch & RM=Buzzard Branch,Main      ,14121.5
1210.794
River Rch & RM=Buzzard Branch,Main      ,12020.3
1245.242
River Rch & RM=Buzzard Branch,Main      ,11709.5
1416.938
River Rch & RM=Buzzard Branch,Main      ,10816.5
1489.443
River Rch & RM=Buzzard Branch,Main      ,9926.8
1591.720
River Rch & RM=Buzzard Branch,Main      ,290.2
1760.950
Boundary for River Rch & Prof#=Buzzard Branch,Main      ,1
Up Type=0
Dn Type=3
Dn Slope=0.039869

--- Buzzard Branch.g01 (geometry) ---

Geom Title=USGS 10m DEM
Program Version=4.00

River Reach=Buzzard Branch  ,Main
Reach XY= 30
     1855916.741      162774.274     1855354.612      162752.488
     1855196.248      162596.323     1854665.372      162400.662
     1854360.511        162445.8     1853931.531      162359.875
     1852586.533       162742.59     1852037.672      162593.244
      1851428.38      162695.694     1850291.347      161591.148
     1849625.996      161334.905     1849294.257      160761.077
     1849309.607      160265.289     1848893.086      159820.999
       1848371.4      159506.096     1848288.095      158596.247
      1848444.47      157756.009     1848016.913      157123.355
     1847776.453      157006.966     1847445.474      156611.722
     1847034.985      156657.206     1846804.569      156521.319
     1846321.285      156033.309     1846148.178       156019.72
     1845631.809      156217.052     1845136.118      155893.287
     1844581.347      155747.947      1844463.52      155607.213
     1845155.615      153859.715     1845022.417      153195.056

Type RM Length L Ch R = 1 ,19045.3 ,390.4,403.4,416.3
XS GIS Cut Line= 4
     1855809.955      162322.779     1855811.356      162515.899
      1855963.71      162988.197     1855978.945      163226.885
#Sta/Elev= 30
     9.7 2259.75    57.9 2254.36   164.2 2246.91   173.8  2245.5   183.5 2242.52
   222.9 2224.65   262.6 2208.17   401.6 2153.65   421.4  2148.6   458.5 2144.22
     471 2143.07     481  2143.8   483.5 2144.72   490.9 2147.43   510.7 2157.41
   520.7 2161.28   530.6 2163.93   540.5 2165.21   570.3 2167.73   600.1 2171.62
     610 2172.03   639.8 2171.72   689.4 2168.08   709.3 2168.84   729.3 2171.94
   739.2 2175.73   749.2 2181.11   818.9 2225.03   888.7 2258.41   928.6 2279.08
#Mann= 3 , 0 , 0
       0      .1       0   458.5    .045       0   483.5      .1       0
Bank Sta=458.5,483.5
XS Rating Curve= 0 ,0
Exp/Cntr=0.3,0.1

Type RM Length L Ch R = 1 ,18641.9 ,275.7,293.8,311.8
XS GIS Cut Line= 4
     1855647.518      162262.287     1855560.938      162512.113
     1855494.645      162956.582     1855507.384      163262.327
#Sta/Elev= 30
     9.8 2230.74    19.6 2226.48    39.2 2221.25      49 2219.89    88.1 2217.31
   107.7 2213.17   146.9 2202.55     235 2174.51   264.4  2167.2   284.4 2165.51
   344.3 2163.13   374.3 2160.62   444.2 2148.76   511.5 2134.26     524 2132.26
     534 2132.76   536.5 2133.72     544 2136.58     564 2149.33     574 2154.16
   603.9 2164.28   643.9 2174.43   653.9  2177.8   723.7 2208.94   743.4 2216.18
   832.2 2242.98   901.3 2261.27   980.3 2275.93  1000.1 2283.38  1019.8    2294
#Mann= 3 , 0 , 0
       0      .1       0   511.5    .045       0   536.5      .1       0
Bank Sta=511.5,536.5
XS Rating Curve= 0 ,0
Exp/Cntr=0.3,0.1

Type RM Length L Ch R = 1 ,18348.1 ,207.6,192.7,177.8
XS GIS Cut Line= 3
     1855553.288      162232.074     1855385.173      162557.096
     1855164.756      162766.306
#Sta/Elev= 30
     9.9 2274.06    69.2 2266.11    98.9 2261.36   148.3 2250.81   187.9 2240.48
   237.4 2225.02   336.3 2188.63   365.9 2174.06   395.3 2160.82   434.5 2141.08
   444.4  2136.5   454.2 2132.95   473.8 2129.79   520.1 2125.36   532.6 2124.92
   542.4 2126.45   571.8 2137.09   620.8 2151.57   650.2 2158.72   689.6 2166.47
   699.5 2169.27   709.3 2173.05   748.9 2191.36   768.6 2199.73   837.8 2224.32
   857.6 2232.62     907 2255.41   916.9 2260.89   926.8 2267.14   976.2 2300.15
#Mann= 3 , 0 , 0
     9.9      .1       0   520.1    .045       0   542.4      .1       0
Bank Sta=520.1,542.4
XS Rating Curve= 0 ,0
Exp/Cntr=0.3,0.1

Type RM Length L Ch R = 1 ,18155.4 ,197.1,193.8,190.5
XS GIS Cut Line= 4
      1855392.73      162147.632     1855169.791       162389.68
     1855048.767      162771.861      1854997.81      163071.237
#Sta/Elev= 30
      10 2374.88    19.9 2374.71    29.9 2373.27    39.9 2369.94    49.9 2365.06
   159.6 2305.01   199.4 2283.97   249.3 2258.04   329.1 2218.69   399.2 2174.28
   469.4 2131.78   479.4 2127.12   489.4 2124.31     507 2121.97   519.5 2120.77
     532 2121.36   539.5 2122.95   569.6 2135.22   589.6 2144.19   599.7 2147.16
   649.8 2156.77   699.9 2164.92   719.9 2168.92   788.7 2186.59   808.3 2192.42
   847.5  2209.2   886.7 2228.37   906.3 2239.45   945.5 2263.19  1033.6 2313.78
#Mann= 3 , 0 , 0
       0      .1       0     507    .045       0     532      .1       0
Bank Sta=507,532
XS Rating Curve= 0 ,0
Exp/Cntr=0.3,0.1

Type RM Length L Ch R = 1 ,17961.6 ,66.5,70.2,73.9
XS GIS Cut Line= 5
     1855138.605      162086.374     1854959.282      162347.887
     1854877.093      162784.985      1854906.98      163039.025
     1854925.659      163102.535
#Sta/Elev= 30
     9.9 2371.26    49.5 2346.03    99.1 2312.28   118.9 2300.95   188.3 2265.94
   277.5 2222.74   327.2 2197.34   357.5 2180.17   448.5 2125.72   458.6  2122.1
   486.5 2116.22     499 2115.63  507.58 2118.13   529.4 2131.87   539.5 2136.96
   559.7 2142.89   600.1 2148.43   620.3 2149.14   650.7 2147.97   660.8 2148.41
   670.9 2150.94   741.6 2182.91   820.9 2210.91   850.4 2223.97   889.7 2247.44
   968.4 2303.75  1017.6 2335.11  1036.6 2343.07    1046  2345.2  1083.8 2347.03
#Mann= 3 , 0 , 0
     9.9      .1       0   486.5    .045       0  507.58      .1       0
Bank Sta=486.5,507.58
XS Rating Curve= 0 ,0
Exp/Cntr=0.3,0.1

Type RM Length L Ch R = 1 ,17891.4 ,121.5,121.2,120.9
XS GIS Cut Line= 4
     1855116.189        162026.6     1854918.187      162321.735
     1854794.903      162695.324     1854787.431      163076.384
#Sta/Elev= 30
     9.9 2392.14    29.6 2385.05    49.4 2374.63    88.9 2349.95   128.3 2323.06
     158  2306.9     306 2234.38   355.4 2208.32   415.9 2173.86   486.5 2129.49
   496.6 2124.09   524.5  2115.3     537 2114.73  544.54 2116.95   567.2 2128.71
   587.4 2136.89   627.8  2145.6     658 2147.29   718.5 2145.05   728.6 2147.15
     809 2185.73   879.2 2208.42   919.3 2225.42   939.4 2236.37   959.4 2249.18
  1029.6 2302.83  1059.7 2323.88  1079.8 2336.27  1099.8 2344.22  1129.9 2345.43
#Mann= 3 , 0 , 0
     9.9      .1       0   524.5    .045       0  544.54      .1       0
Bank Sta=524.5,544.54
XS Rating Curve= 0 ,0
Exp/Cntr=0.3,0.1

Type RM Length L Ch R = 1 ,17770.2 ,174.1,168.8,163.7
XS GIS Cut Line= 4
      1854991.44      162039.347     1854814.422      162247.029
     1854675.355      162684.116     1854564.671      162988.431
#Sta/Elev= 30
    10.1 2355.71    20.2 2351.77    60.6 2331.58   131.4 2301.23   202.1 2265.83
   222.4 2253.98   252.7  2233.3   272.9 2221.12   372.6 2171.43   382.6 2165.43
   412.5 2143.65   432.4 2130.58   452.4 2119.01   462.3 2114.51   472.3 2112.47
   484.8 2114.93   502.2 2124.15   512.2 2128.27   552.1 2135.22     582 2141.72
   601.9 2142.97   631.9 2140.79   661.8  2140.4   691.7 2141.49   701.6 2143.21
   751.2 2157.04   829.7 2184.84   849.3  2190.9   927.8 2208.29  1055.4 2242.09
#Mann= 3 , 0 , 0
    10.1      .1       0   462.3    .045       0   484.8      .1       0
Bank Sta=462.3,484.8
XS Rating Curve= 0 ,0
Exp/Cntr=0.3,0.1

Type RM Length L Ch R = 1 ,17601.5 ,164.9,163.4,161.8
XS GIS Cut Line= 4
     1854869.621      161936.939     1854611.845      162228.338
     1854559.542       162680.38      1854570.75      162867.175
#Sta/Elev= 30
      10 2278.77    69.8 2294.23    89.8 2298.15   119.7 2302.48   129.7 2303.17
   139.7 2302.42   149.6 2298.08   159.6 2291.83   179.6 2275.99   189.5 2269.26
   209.5 2260.01   229.4 2253.95   309.2 2236.91   329.2 2230.36   389.1 2198.53
   480.1 2141.42   520.5  2121.5   548.5 2110.39     561 2108.88   571.1 2111.36
   591.3 2119.69   601.4 2121.03     652 2118.21   672.2 2119.59   682.3 2121.44
   773.3 2149.39   823.9 2156.56   942.6 2179.83   991.8 2190.72  1031.2 2201.89
#Mann= 3 , 0 , 0
      10      .1       0   548.5    .045       0   571.1      .1       0
Bank Sta=548.5,571.1
XS Rating Curve= 0 ,0
Exp/Cntr=0.3,0.1

Type RM Length L Ch R = 1 ,17438   ,302.4,305.1,307.9
XS GIS Cut Line= 4
     1854705.242      161940.675     1854451.201      162243.282
     1854428.786       162635.55     1854522.183        162953.1
#Sta/Elev= 30
     9.9 2226.72    49.4 2231.62    59.3 2231.11    98.8 2220.39   177.8 2204.85
   217.3 2199.82   237.1 2199.97   286.5 2204.87   316.1 2201.74   335.8  2195.2
   355.6 2186.75   395.1 2168.48   445.5 2142.25   465.6 2133.71   485.8  2127.6
   505.9 2123.25   546.2 2121.15   556.3 2119.19   566.4 2115.14  588.91 2101.27
   596.6 2098.66   609.1 2100.78   667.1 2131.94   687.3 2139.96   747.7  2147.3
     798  2159.4   878.3 2176.32   968.6 2201.23  1078.9  2221.4    1119 2230.62
#Mann= 3 , 0 , 0
     9.9      .1       0  588.91    .045       0   609.1      .1       0
Bank Sta=588.91,609.1
XS Rating Curve= 0 ,0
Exp/Cntr=0.3,0.1

Type RM Length L Ch R = 1 ,17132.9 ,298.8,287.6,276.5
XS GIS Cut Line= 4
     1854458.673       161963.09     1854167.274      162232.074
     1854099.684      162657.207     1854195.229       163001.17
#Sta/Elev= 30
     9.9 2139.88    69.4 2135.22     119 2140.34   158.6 2129.97     228 2121.45
   356.9 2118.69   396.6 2118.57   416.6 2120.19   436.6 2119.19   506.7 2106.26
   546.7 2088.37   574.3 2081.03   586.8 2080.49   599.3  2080.5   636.8 2081.58
   646.8 2085.49   686.9 2114.46   706.9 2127.26   736.9 2143.88     777 2161.78
     827  2179.9   916.3 2201.83   936.1 2208.95   985.7 2235.47  1045.2 2274.31
  1124.5 2321.93  1134.4 2326.97  1144.4 2329.86  1164.2 2332.41    1184 2339.44
#Mann= 3 , 0 , 0
     9.9      .1       0   574.3    .045       0   599.3      .1       0
#XS Ineff= 2 , 0
                           638.6         2103.87
Permanent Ineff=
       F       F
Bank Sta=574.3,599.3
XS Rating Curve= 0 ,0
Exp/Cntr=0.3,0.1

Type RM Length L Ch R = 1 ,16845.2 ,297.4,296.7,296
XS GIS Cut Line= 4
     1853820.062      161831.191     1853807.322      162168.785
     1853931.315      162666.369      1854055.74       162888.56
#Sta/Elev= 30
     9.9  2313.6    59.6 2307.82    99.4 2304.33   109.3 2301.98   129.2    2294
     159 2279.98   228.5 2244.16     368    2175   418.3 2148.34   488.7 2107.15
   518.8 2091.02   528.9 2084.41   536.5 2081.25   538.9 2080.26     549 2078.99
   561.5 2079.46   579.2  2081.8   599.3 2087.07   669.6 2118.54   719.9 2147.97
   770.2  2171.8   780.2 2177.17   820.5 2203.09   850.6 2223.67   870.2 2235.53
   909.4 2256.37   938.8 2269.66   958.4 2276.55   987.8 2281.75  1105.3 2291.63
#Mann= 3 , 0 , 0
       0      .1       0   536.5    .045       0   561.5      .1       0
Bank Sta=536.5,561.5
XS Rating Curve= 0 ,0
Exp/Cntr=0.3,0.1

Type RM Length L Ch R = 1 ,16548.5 ,303.9,302.5,301
XS GIS Cut Line= 4
     1853532.174      161895.844     1853520.966      162265.697
     1853629.307      162657.965     1853812.365      162915.741
#Sta/Elev= 30
      10 2338.35      40 2321.08      90 2290.34     130 2267.29     160 2251.32
     240 2212.13     310 2179.95   409.7 2140.87   479.2 2109.97   528.8    2090
   538.8 2085.53   548.7 2080.09     556 2077.15   558.6  2076.1   568.5 2074.96
     581 2076.27   598.3 2080.36   618.2 2083.21   628.1 2085.74     638 2090.51
   687.6 2118.52   707.5 2127.75   767.1 2153.19   826.4 2191.46   865.9 2215.31
   915.3 2246.19   944.9    2263    1024 2305.05  1053.6  2324.6  1093.1 2353.21
#Mann= 3 , 0 , 0
       0      .1       0     556    .045       0     581      .1       0
Bank Sta=556,581
XS Rating Curve= 0 ,0
Exp/Cntr=0.3,0.1

Type RM Length L Ch R = 1 ,16246.1 ,334.5,334,333.5
XS GIS Cut Line= 4
     1853182.143      161990.297     1853213.991       162327.89
     1853366.864      162786.508     1853519.736      163028.556
#Sta/Elev= 30
      10  2340.1    19.9 2339.03    39.9 2335.03    69.8 2333.33    79.8 2331.08
    89.8 2327.44   139.6 2304.32   159.6 2292.83   209.4 2256.94   229.4 2244.39
   319.1 2197.31   389.4 2155.87   459.9 2116.03   500.2 2093.64   538.1 2073.96
   540.5 2072.78   550.6 2071.59   563.1 2072.75   590.9 2078.63   621.1 2080.51
   631.2 2083.13   701.7 2114.28   762.1 2135.92   772.2  2138.9   822.5 2150.39
   950.9 2192.98   990.3 2208.49  1029.8 2227.65  1069.3 2250.06  1108.8  2274.6
#Mann= 3 , 0 , 0
       0      .1       0   538.1    .045       0   563.1      .1       0
Bank Sta=538.1,563.1
XS Rating Curve= 0 ,0
Exp/Cntr=0.3,0.1

Type RM Length L Ch R = 1 ,15912.1 ,219.8,219.6,219.3
XS GIS Cut Line= 4
     1852832.116      162026.608     1852889.443      162421.529
      1853026.28      162806.935     1853188.818      163115.825
#Sta/Elev= 30
      10 2148.78   159.6 2155.12   279.3 2147.83   389.1 2138.93     419 2133.04
   478.9 2115.27   508.8  2109.5   558.7  2097.6   568.6 2093.63   578.6 2086.24
   588.6 2076.23     596 2071.21   598.6 2069.45   608.5 2068.04     621 2068.94
   648.4 2072.46   688.3 2073.49   698.3 2076.71   738.2 2102.87   748.2 2108.18
   758.2 2111.24   788.1 2114.45     838 2123.29   867.9 2131.77   887.8 2139.11
   947.7 2167.76  1047.4 2211.16  1077.3 2225.62  1107.2 2243.62  1157.1 2277.73
#Mann= 3 , 0 , 0
       0      .1       0     596    .045       0     621      .1       0
Bank Sta=596,621
XS Rating Curve= 0 ,0
Exp/Cntr=0.3,0.1

Type RM Length L Ch R = 1 ,15692.5 ,296.4,315.2,334
XS GIS Cut Line= 4
     1852577.328      162115.784     1852679.295      162490.019
     1852814.703       162862.39     1852900.809       163143.63
#Sta/Elev= 30
     9.9 2246.31   139.2 2192.02   238.7 2152.98   308.3 2123.85   338.2 2112.45
   387.9 2096.36   417.6 2089.84   457.2 2089.29   516.7 2084.63   536.5 2081.02
   566.2  2074.6   593.3 2067.32   605.8 2065.36   618.3 2065.57   655.3 2068.65
     685 2070.22   724.7 2069.32   734.6 2071.21   744.5 2075.17   803.7 2106.04
   882.1  2152.4   921.4 2174.08   960.6 2198.71   970.4 2203.53   980.2 2207.06
   999.8 2212.56  1009.6 2216.05  1019.4 2220.52    1039 2230.69  1078.2 2254.48
#Mann= 3 , 0 , 0
       0      .1       0   593.3    .045       0   618.3      .1       0
Bank Sta=593.3,618.3
XS Rating Curve= 0 ,0
Exp/Cntr=0.3,0.1

Type RM Length L Ch R = 1 ,15377.3 ,178,177.3,176.5
XS GIS Cut Line= 4
     1852514.872       162187.77     1852478.602      162642.353
     1852410.898       162838.21     1852447.168      163174.311
#Sta/Elev= 30
     9.9 2260.95    99.1 2231.83   168.5 2206.77   188.4  2198.9   198.3 2195.69
   208.2 2193.56   257.8 2186.14   267.7 2183.74   277.6 2180.55   297.4 2173.28
   327.1 2161.17   386.6 2132.65   436.2 2110.63   515.2 2074.41     535 2063.86
   542.2 2060.91   544.8 2059.84   554.7 2058.21   567.2 2058.72     604 2063.46
   623.8 2066.64   673.2 2078.95     713 2093.93   742.8 2102.03   792.5 2120.45
   832.3 2134.29   852.2 2142.52     882 2155.87   921.8 2174.69  1001.3 2217.22
#Mann= 3 , 0 , 0
       0      .1       0   542.2    .045       0   567.2      .1       0
Bank Sta=542.2,567.2
XS Rating Curve= 0 ,0
Exp/Cntr=0.3,0.1

Type RM Length L Ch R = 1 ,15200   ,64.6,65,65.3
XS GIS Cut Line= 4
     1852351.634      162134.941     1852362.841      162411.397
      1852209.67      162897.062     1852265.708      163274.386
#Sta/Elev= 30
     9.9 2262.11    69.2 2251.63    98.8 2245.33   148.2 2232.59     168 2225.92
   197.6 2213.24   276.7 2183.31   406.5 2129.02   466.4 2103.27   496.4 2087.86
   516.3 2076.25   543.8 2059.14   546.3 2057.72   556.3 2056.09   568.8 2056.73
   596.2 2059.68   606.2 2061.48   656.1 2073.63   666.1 2077.16     726 2102.77
     806 2140.52   846.2 2160.88   876.3  2177.8   936.5 2215.73   996.7 2249.44
  1016.8 2258.95  1036.9  2267.5  1117.2 2295.86  1137.3 2305.02  1167.4 2320.33
#Mann= 3 , 0 , 0
       0      .1       0   543.8    .045       0   568.8      .1       0
Bank Sta=543.8,568.8
XS Rating Curve= 0 ,0
Exp/Cntr=0.3,0.1

Type RM Length L Ch R = 1 ,15135.1 ,93.1,87.2,81
XS GIS Cut Line= 4
      1852309.76      162112.956      1852255.98      162540.034
     1852180.055      162770.973     1852199.036         163081.
#Sta/Elev= 30
      10 2241.16    50.1 2230.71   100.1 2216.82   150.2 2201.38   190.2 2188.21
   320.3 2141.67   370.4 2124.49   420.4 2108.11   430.5 2103.89   440.2 2098.67
   449.9 2094.23   498.5 2079.47     518 2070.81   537.4  2059.9   544.4 2057.06
   547.1 2055.97   556.9 2054.85   569.4 2055.81   595.8 2058.24   605.5 2060.05
   644.4 2070.02   703.7 2089.55   743.8 2105.79     774 2119.75   834.2 2149.52
   854.3 2161.35   894.4 2186.15   931.6 2207.64   967.7 2227.33   985.8 2235.93
#Mann= 3 , 0 , 0
       0      .1       0   544.4    .045       0   569.4      .1       0
Bank Sta=544.4,569.4
XS Rating Curve= 0 ,0
Exp/Cntr=0.3,0.1

Type RM Length L Ch R = 1 ,15047.9 ,114.9,108.1,101.1
XS GIS Cut Line= 4
     1852252.817      162128.773     1852145.256      162540.034
     1852119.948      162774.136     1852151.583      163074.673
#Sta/Elev= 30
     9.9 2205.63      89 2180.01   168.1 2152.65   207.6 2137.95   296.6 2103.17
   326.2 2092.52   365.8 2079.54   375.7  2075.9   395.4 2066.78   405.3 2062.65
   415.2 2059.74   425.1 2058.14   474.1 2056.99   493.8 2055.62   510.7  2053.7
   523.2 2053.18   535.7 2054.07   562.4 2056.84   572.3 2058.25   591.9 2062.37
   611.5 2067.26   700.9 2097.53     721 2104.87   731.1 2109.01   781.4 2132.79
   811.7  2148.5     852 2171.62   932.5 2218.95   952.7 2229.96   962.8 2234.51
#Mann= 3 , 0 , 0
       0      .1       0   510.7    .045       0   535.7      .1       0
Bank Sta=510.7,535.7
XS Rating Curve= 0 ,0
Exp/Cntr=0.3,0.1

Type RM Length L Ch R = 1 ,14939.8 ,84.9,85.3,86.2
XS GIS Cut Line= 4
     1852183.219      162056.012     1852021.878      162502.072
     1852056.677      162761.482     1852110.457      162986.094
#Sta/Elev= 30
    10.1 2175.45   100.9 2143.74   151.4 2126.66   201.8 2110.14   232.1 2101.86
   242.2  2099.6   272.5 2094.48   353.2 2087.63   403.7 2081.43   454.2 2077.36
   474.3 2074.88   504.5 2062.43   534.7 2052.13   544.8 2049.95   562.5 2048.56
     575 2048.35   587.5 2049.58   615.3 2055.07   635.4  2056.9   655.5 2057.89
   685.7 2061.75   695.8 2063.98   705.9 2066.99   736.1 2077.46   796.3  2100.2
   816.4  2108.5   836.5 2117.59   876.7 2136.74   906.8 2152.04     967 2185.86
#Mann= 3 , 0 , 0
       0      .1       0   562.5    .045       0   587.5      .1       0
Bank Sta=562.5,587.5
XS Rating Curve= 0 ,0
Exp/Cntr=0.3,0.1

Type RM Length L Ch R = 1 ,14854.5 ,168.2,169.1,170.1
XS GIS Cut Line= 4
     1852105.065      162022.864     1851929.478      162433.812
     1851970.573      162781.249      1852146.16      163177.253
#Sta/Elev= 30
     9.9 2151.76     139 2152.24   218.5 2157.09   278.1 2157.59   307.9    2156
   337.6 2152.99   417.1 2138.45   446.9 2135.06   476.9 2122.25   506.9 2106.82
   556.8  2079.3   586.8 2059.76   606.8  2049.5   614.3 2047.14   626.8 2045.58
   639.3 2047.01   696.8 2055.66   736.8 2059.49   776.8 2071.82   816.9 2087.46
   847.1 2101.64   897.5 2128.49   978.1 2166.31  1028.5 2192.01  1088.9 2224.72
    1109 2233.65  1159.4 2248.85  1179.6 2257.21  1199.7 2267.92  1229.9 2287.62
#Mann= 3 , 0 , 0
       0      .1       0   614.3    .045       0   639.3      .1       0
Bank Sta=614.3,639.3
XS Rating Curve= 0 ,0
Exp/Cntr=0.3,0.1

Type RM Length L Ch R = 1 ,14685.3 ,270.4,269.2,267.9
XS GIS Cut Line= 4
     1851883.776       162163.59     1851772.548      162461.003
     1851799.146      162782.596     1851898.284      163065.501
#Sta/Elev= 30
     9.9 2248.36    59.5 2248.54    89.3 2245.08   109.2 2243.76     129 2239.75
   158.8 2231.23   168.7 2227.32   188.5 2215.95   208.4 2207.77   248.1 2185.13
   297.7 2161.35   317.5 2150.88     368  2117.4   398.2 2096.23   418.4 2081.23
   448.6 2056.13   458.7 2049.99   468.8 2046.48   496.6 2041.03   509.1 2039.84
   521.6 2040.92   559.5 2047.91   569.6 2050.53   680.2 2092.46   720.2  2109.4
   770.1 2133.71   800.1 2150.05     870 2192.59     910 2218.02     940  2238.3
#Mann= 3 , 0 , 0
       0      .1       0   496.6    .045       0   521.6      .1       0
Bank Sta=496.6,521.6
XS Rating Curve= 0 ,0
Exp/Cntr=0.3,0.1

Type RM Length L Ch R = 1 ,14416.2 ,262.7,294.7,326.7
XS GIS Cut Line= 4
     1851787.487      162090.305      1851492.38      162448.755
      1851555.89      162930.685     1851634.615      163319.655
#Sta/Elev= 30
    10.1 2309.51    60.6 2316.57    80.7 2317.13    90.8 2315.18   100.9 2311.72
   141.3  2294.8   171.6  2279.3   201.9  2260.9   222.1 2252.26   242.2 2241.61
     434 2109.61   444.1 2102.05   464.3 2084.37   523.8 2066.88   603.2 2037.51
   613.1 2035.39     623 2034.55   699.8 2030.29   712.3 2030.08   724.8 2031.22
   742.1 2035.15     752 2038.76     871 2092.18     881 2095.87   900.8 2099.85
   920.6 2102.58  1039.7 2110.76  1158.7 2116.81    1258 2114.76  1347.3 2105.06
#Mann= 3 , 0 , 0
       0     .08       0   699.8    .045       0   724.8     .08       0
Bank Sta=699.8,724.8
XS Rating Curve= 0 ,0
Exp/Cntr=0.3,0.1

Type RM Length L Ch R = 1 ,14121.5 ,476.8,466.4,456.1
XS GIS Cut Line= 4
     1851554.425      162175.626     1851458.757      162474.907
     1851074.082      162708.165     1850895.731      162931.104
#Sta/Elev= 30
     9.8 2201.39    39.3 2185.67    68.7 2167.98    78.5 2162.91     108  2151.9
   186.6 2116.69     216 2102.59   255.3 2081.39   265.1 2077.18   314.2 2061.46
   364.2 2041.45   394.2 2034.71   444.2 2029.24   521.6 2022.93   534.1  2021.8
   546.6 2022.25   594.1 2032.12   644.1 2050.62   654.1 2055.23   664.1 2061.13
   694.1 2084.38   704.1 2091.12   724.1 2101.28   773.9 2121.72   813.3 2134.95
   882.2 2155.32   911.7  2165.7   931.4 2174.05   990.5  2202.3  1049.6 2226.34
#Mann= 3 , 0 , 0
       0     .08       0   521.6    .045       0   546.6     .08       0
Bank Sta=521.6,546.6
XS Rating Curve= 0 ,0
Exp/Cntr=0.3,0.1

Type RM Length L Ch R = 1 ,13655   ,448.5,452.5,456.6
XS GIS Cut Line= 4
     1851481.742      161848.257     1851138.523      162020.831
     1850806.555      162453.377     1850660.052      162733.643
#Sta/Elev= 30
    10.1 2329.24    50.5  2314.6    70.8 2309.44      91 2306.03   131.4 2302.36
   161.8 2294.16   222.4 2269.65   303.3  2231.6   384.2 2190.07     475 2132.91
   545.7 2086.93   626.5  2036.6   646.7 2022.48   656.8 2017.62   666.9  2016.2
   679.4 2016.43   737.6  2016.8   798.1 2019.07   808.2 2022.36   838.5 2039.14
   878.9 2050.05   919.3 2065.35   939.3 2074.89   998.6 2106.29  1028.2 2118.19
  1067.8 2132.21    1137 2153.58  1206.1 2167.58  1225.9 2174.11  1245.7  2182.2
#Mann= 3 , 0 , 0
    10.1     .08       0   656.8    .045       0   679.4     .08       0
#XS Ineff= 2 , 0
                          763.66         2029.02
Permanent Ineff=
       F       F
Bank Sta=656.8,679.4
XS Rating Curve= 0 ,0
Exp/Cntr=0.3,0.1

Type RM Length L Ch R = 1 ,13202.5 ,317.6,316.5,315.5
XS GIS Cut Line= 4
     1851131.409      161561.621     1850802.059      161780.162
     1850456.222      162115.784      1850296.98      162370.571
#Sta/Elev= 30
     9.9 2197.76    49.4 2185.39   108.7  2178.4   138.3 2174.09   207.5 2166.48
   256.9 2159.16   286.6 2152.83   326.1  2141.9   365.6 2127.92   525.8 2062.99
   596.1 2029.72   606.1 2022.39   616.1 2013.21   623.7 2007.74   626.2 2005.94
   636.2 2005.17   648.7 2006.36   686.4 2009.85   716.5 2013.71   756.7 2015.13
   776.8 2017.03   796.9 2020.94     827 2031.02   847.1 2039.33   867.1 2048.77
  1017.4  2124.1  1077.5 2160.55  1107.5 2175.77  1127.6 2187.02  1177.6  2217.6
#Mann= 3 , 0 , 0
       0      .1       0   623.7    .045       0   648.7     .08       0
Bank Sta=623.7,648.7
XS Rating Curve= 0 ,0
Exp/Cntr=0.3,0.1

Type RM Length L Ch R = 1 ,12886   ,864.7,865.7,866.6
XS GIS Cut Line= 4
     1850887.643       161334.33     1850644.334      161477.425
     1850244.304      161894.862      1850116.91      162187.868
#Sta/Elev= 30
    10.1 2203.14    60.5 2195.25   110.9 2189.24     121 2186.66   131.1  2182.5
   171.4 2161.67   201.6 2144.01   241.9 2118.67   262.1 2107.45   282.3 2097.42
   312.2 2084.39   322.1 2080.58     362 2071.18   491.6 2031.49   598.7 2000.59
   611.2 1999.41   623.7 2000.04     671 2004.98   720.9 2012.16   740.8 2016.41
   770.7 2025.97   790.7 2034.26   810.6 2044.65   850.5 2069.41   870.4 2080.53
   980.2 2132.66  1040.2 2163.36  1100.1  2195.5    1120 2200.55  1179.9 2203.49
#Mann= 3 , 0 , 0
       0      .1       0   598.7    .045       0   623.7      .1       0
Bank Sta=598.7,623.7
XS Rating Curve= 0 ,0
Exp/Cntr=0.3,0.1

Type RM Length L Ch R = 1 ,12020.3 ,305.6,310.9,316.1
XS GIS Cut Line= 4
     1850207.805      161026.567      1849848.59      161148.667
     1849478.737      161525.992     1849303.309      161752.712
#Sta/Elev= 30
      10 2261.35    49.9 2233.94    69.9 2222.62    79.9 2218.04   109.8 2206.99
   199.7 2177.44   269.6 2155.45   309.5  2140.3   349.4 2122.86   379.4 2111.45
   439.2 2072.52   469.1 2051.77     499 2032.98   528.9 2010.96   538.9 2006.01
   588.7 1995.02   648.6  1985.2   698.4 1986.07   775.6 1984.89   788.1 1984.77
   798.1 1985.57   800.6 1986.43   808.1    1989     828 2000.92   897.8 2036.76
     977  2073.8  1046.1 2108.01  1065.9 2118.94  1135.1  2160.6  1194.4 2193.94
#Mann= 3 , 0 , 0
      10      .1       0   775.6    .045       0   800.6     .08       0
#XS Ineff= 2 , 0
          760.48 2035.85
Permanent Ineff=
       F       F
Bank Sta=775.6,800.6
XS Rating Curve= 0 ,0
Exp/Cntr=0.3,0.1

Type RM Length L Ch R = 1 ,11709.5 ,284,291.3,298.6
XS GIS Cut Line= 4
     1850201.435      160816.368     1849768.296      160905.543
     1849261.604      161244.291     1848984.825      161612.578
#Sta/Elev= 30
    10.1  2356.2    80.4 2347.52   150.8 2344.77   170.9 2341.35     191 2334.74
   271.4 2289.07   291.5  2274.7   311.6 2258.63   341.7 2229.14     402 2182.72
   502.2 2119.91   552.1 2089.69   602.1 2062.69     682 2024.12     712 2012.38
     762 1995.76   791.9 1982.67   799.4 1980.36   811.9 1979.01   824.4 1980.51
   861.9 1986.51   951.8 2019.59   971.8 2025.59  1011.8 2033.06  1131.8 2062.07
    1242 2085.84  1352.2 2117.41  1382.2 2126.85  1402.3 2134.45  1512.4 2180.52
#Mann= 3 , 0 , 0
       0      .1       0   799.4    .045       0   824.4      .1       0
Bank Sta=799.4,824.4
XS Rating Curve= 0 ,0
Exp/Cntr=0.3,0.1

Type RM Length L Ch R = 1 ,11418.2 ,213.6,221.2,228.8
XS GIS Cut Line= 4
     1849959.387      160720.822     1849612.883      160755.952
        1849074.      160937.392     1848710.928      161281.355
#Sta/Elev= 30
      10 2286.36    39.8 2286.49    59.7  2281.5    69.7 2276.43   149.3 2229.74
   318.4 2116.84   428.1 2051.33   497.9 2022.15   527.8 2012.13   597.7 1994.68
   617.6 1987.04     635 1978.03   647.5 1974.88     660  1975.8   717.4 1985.09
   787.2 2002.91     877 2042.32   976.9 2090.67  1006.9 2102.91  1036.9 2110.54
  1106.9 2120.67  1126.9 2126.44  1146.9 2139.65    1187 2175.45    1197 2182.62
    1217 2193.56    1277 2221.34    1297  2232.6    1377  2284.6    1417 2315.21
#Mann= 3 , 0 , 0
       0      .1       0     635    .045       0     660      .1       0
Bank Sta=635,660
XS Rating Curve= 0 ,0
Exp/Cntr=0.3,0.1

Type RM Length L Ch R = 1 ,11197   ,140.6,142.4,144.2
XS GIS Cut Line= 4
     1850020.441      160416.433     1849467.529      160629.379
     1849097.677      160648.058     1848701.673      161014.175
#Sta/Elev= 30
      10 2124.82    30.1 2122.31    40.2 2123.27   100.4 2136.19   170.7 2147.94
   291.2 2158.21   311.3 2158.42   321.4 2156.93   421.8 2127.81     472 2110.85
   492.1 2099.23   532.2 2068.97   552.3 2059.29   672.6 2012.55   712.6 1994.99
   780.2 1972.81   792.7 1970.75   805.2 1971.88   852.7    1982   932.8 2009.48
   942.8 2014.55   962.8 2027.19  1042.7 2066.92  1112.6 2103.42  1162.6 2127.67
  1262.4 2179.37  1332.4  2212.2  1392.3 2246.76  1422.2 2258.52  1502.1 2286.83
#Mann= 3 , 0 , 0
       0      .1       0   780.2    .045       0   805.2     .08       0
Bank Sta=780.2,805.2
XS Rating Curve= 0 ,0
Exp/Cntr=0.3,0.1

Type RM Length L Ch R = 1 ,11054.6 ,252.3,238.1,223
XS GIS Cut Line= 4
     1850004.996      160267.884     1849485.127      160500.012
     1849153.862      160495.176     1848984.603      160599.149
#Sta/Elev= 30
      10 2068.73   119.9 2070.28   189.8 2078.31   399.5 2094.16   429.5 2093.51
   459.5 2090.16   489.4 2084.27   509.4 2077.22   529.4 2067.07   559.3  2047.4
   579.4 2036.69   599.5 2029.87   639.6 2023.46   649.7 2020.26   689.8 2000.78
   760.1 1970.33   767.7 1968.58   780.2 1967.99   792.7  1969.3   840.4 1973.95
   860.5 1977.48   900.6  1994.8   950.3  2013.3   970.2 2022.71     990 2033.86
  1009.9 2043.22  1049.6 2056.09  1069.5 2064.13  1089.4 2074.87  1099.3 2081.83
#Mann= 3 , 0 , 0
       0      .1       0   767.7    .045       0   792.7     .08       0
Bank Sta=767.7,792.7
XS Rating Curve= 0 ,0
Exp/Cntr=0.3,0.1

Type RM Length L Ch R = 1 ,10816.5 ,367.2,357.4,348.5
XS GIS Cut Line= 4
     1849946.647      160077.484     1849587.078       160128.77
      1849004.28      160416.433      1848882.91      160657.125
#Sta/Elev= 30
    10.1 2075.37    80.7 2068.35   141.2 2063.78   211.9    2060   272.4 2058.13
   363.2 2044.66   503.2 2009.22   553.2 1999.59   593.2  1994.6   623.2 1987.89
   643.2 1980.55   673.2 1965.39   680.7 1963.69   693.2 1963.09   705.7 1963.65
   793.2 1969.43   803.2 1970.69   813.2 1973.53   893.1 2012.73   903.1 2016.21
   913.1 2018.27   933.1 2020.32   943.1  2022.8  1013.1  2054.1    1073 2071.57
    1103 2082.17  1132.9 2094.73  1252.7 2150.09  1262.7 2154.01  1282.7 2160.19
#Mann= 3 , 0 , 0
       0      .1       0   680.7    .045       0   705.7     .08       0
Bank Sta=680.7,705.7
XS Rating Curve= 0 ,0
Exp/Cntr=0.3,0.1

Type RM Length L Ch R = 1 ,10459.1 ,534.7,532.2,529.1
XS GIS Cut Line= 4
     1849583.575      159657.084       1849284.2      159784.478
      1848870.17      160223.987     1848788.407      160430.772
#Sta/Elev= 30
     9.9 2252.71    19.7 2245.62    39.4 2234.56   177.5 2166.23     207 2148.98
   266.2 2110.47   285.9 2099.03   315.5 2084.41   375.7 2062.35   405.9 2053.91
   466.2 2039.58   506.5 2025.96   546.8 2007.59   597.1 1976.74   617.2 1966.57
   637.3 1961.63   675.1 1958.26   687.6  1957.4   700.1 1958.12   727.9 1962.63
   788.3 1967.97   808.4 1974.15   828.5 1983.36   888.9 2014.18   939.3  2035.5
   979.7 2055.92  1080.8 2104.27  1121.2 2125.59  1131.3    2130  1151.5 2135.81
#Mann= 3 , 0 , 0
       0      .1       0   675.1    .045       0   700.1     .08       0
Bank Sta=675.1,700.1
XS Rating Curve= 0 ,0
Exp/Cntr=0.3,0.1

Type RM Length L Ch R = 1 ,9926.8  ,304.9,312.6,320.3
XS GIS Cut Line= 4
     1848990.196      159382.235     1848857.421      159479.595
     1848519.782      159887.222     1848441.021      160133.148
#Sta/Elev= 30
     9.7 2082.74    67.8 2068.17   116.2 2057.48   135.6 2055.87   164.6 2055.84
   204.6 2048.24   234.6 2037.16   244.5 2034.58   284.5 2029.43   294.5 2025.92
   304.5 2018.94   324.4  2002.6   354.4 1980.21   374.4 1967.19   394.3 1957.82
   421.8 1949.45   434.3 1947.22   446.8 1947.66   494.2 1951.38   574.1 1960.85
   614.1  1967.1     654 1972.08   703.9 1983.62   733.7 1995.04   813.1 2031.36
   852.9 2050.55   882.7 2063.44   902.5 2073.42   932.3 2090.69   952.2  2099.4
#Mann= 3 , 0 , 0
       0      .1       0   421.8    .045       0   446.8     .08       0
Bank Sta=421.8,446.8
XS Rating Curve= 0 ,0
Exp/Cntr=0.3,0.1

Type RM Length L Ch R = 1 ,9614.3  ,449.5,465.1,480.8
XS GIS Cut Line= 4
     1848978.128      159280.724     1848727.824      159336.762
     1848208.536      159699.143     1848219.744      159912.089
#Sta/Elev= 30
     9.9 2108.87    29.6 2105.07    49.3 2103.96   108.5 2112.75   138.1 2114.85
   157.8 2121.15   167.7 2119.95   256.5 2077.58   306.8 2056.81   367.1 2028.51
   457.5 1991.65     558 1952.95   578.1 1946.57     636 1942.23   648.5 1941.88
     661 1944.77   668.6 1948.88   688.7 1967.04   698.8 1974.39   708.8 1981.06
   718.9 1985.51   789.2 1992.92   819.4 2001.43   829.4 2007.71   859.6 2036.57
   869.6 2043.41   899.4 2055.56   928.5 2060.93   986.7 2065.51    1103 2068.12
#Mann= 3 , 0 , 0
       0     .08       0     636    .045       0     661     .08       0
Bank Sta=636,661
XS Rating Curve= 0 ,0
Exp/Cntr=0.3,0.1

Type RM Length L Ch R = 1 ,9149.1  ,455.6,457.5,459.4
XS GIS Cut Line= 4
     1848952.976      158962.788     1848602.643      159096.552
     1848093.068      159122.031     1847685.408      159300.382
#Sta/Elev= 30
     9.9 2150.76    59.2 2147.07     148  2135.6   177.6 2133.25   187.5 2130.39
   197.4 2125.13   236.8 2097.93   286.2 2069.75   365.1 2029.56     455 1987.76
     475 1982.99   505.1 1981.52   615.1 1938.43   642.6 1933.62   655.1 1932.74
   667.6 1935.09   765.2 1980.22   795.2 1999.56   815.2 2010.29   865.2 2030.52
   905.4 2051.12   925.7 2063.77   966.1 2101.66   976.2 2109.04   996.5 2118.79
  1026.8 2126.77  1067.2 2133.22  1208.8  2144.5  1269.5 2167.59  1330.2 2201.74
#Mann= 3 , 0 , 0
       0     .08       0   642.6    .045       0   667.6     .08       0
Bank Sta=642.6,667.6
XS Rating Curve= 0 ,0
Exp/Cntr=0.3,0.1

Type RM Length L Ch R = 1 ,8691.6  ,453.9,458.7,463.5
XS GIS Cut Line= 4
     1848819.213      158739.849     1848653.504      158663.509
     1848016.632      158650.674     1847710.887       158720.74
#Sta/Elev= 30
     9.6 2128.24    38.4 2111.97   134.4 2061.02   182.4 2036.68   303.8 1986.81
   313.9 1984.52   374.6 1981.18   384.7 1979.81   394.8 1976.04   455.4 1945.07
   465.6 1940.69   485.8 1935.74   533.9 1926.79   546.4 1925.31   556.6 1926.24
   558.9 1927.41   566.7 1931.35     688 2020.94   708.2 2034.54   738.6 2053.19
   809.3 2093.74   907.7 2141.29   946.9 2162.21   956.7 2168.05   976.3 2181.61
  1015.5 2212.22  1025.3 2219.12  1044.9 2230.87  1054.7 2235.62  1133.1 2262.76
#Mann= 3 , 0 , 0
       0     .08       0   533.9    .045       0   558.9     .08       0
Bank Sta=533.9,558.9
XS Rating Curve= 0 ,0
Exp/Cntr=0.3,0.1

Type RM Length L Ch R = 1 ,8233    ,446.9,437.9,428.9
XS GIS Cut Line= 4
      1848882.91      158421.365     1848708.669      158275.808
     1848124.917      158160.208     1847812.802      158204.796
#Sta/Elev= 30
     9.9 2153.54   118.5  2093.6   128.3  2090.5   167.8 2089.46   177.7  2085.2
   187.6 2077.61   217.2    2051   257.3 2025.93   287.6 2010.55   358.2 1978.25
   418.7    1949   448.9 1936.78   479.2 1927.69   499.4  1924.2   519.5 1923.26
   537.3 1920.51   549.8 1918.51   559.9 1920.17   562.3 1921.72     570  1926.7
   590.1 1943.61   630.5 1969.43   822.1 2072.43   891.1 2105.38   950.2  2138.4
   969.9 2148.43    1029 2173.38  1058.6 2184.63  1088.1 2193.52  1137.4 2205.84
#Mann= 3 , 0 , 0
       0     .08       0   537.3    .045       0   562.3     .08       0
Bank Sta=537.3,562.3
XS Rating Curve= 0 ,0
Exp/Cntr=0.3,0.1

Type RM Length L Ch R = 1 ,7795    ,475.1,459,443
XS GIS Cut Line= 4
     1849061.261      157816.245     1848671.117      157751.426
     1848182.244      157816.245     1847742.736      158013.705
#Sta/Elev= 30
     9.9 2081.96    39.5 2066.72    69.2 2053.92   108.8 2039.05   138.4 2030.95
   158.2 2028.45   197.7 2027.41   257.1 2022.19   355.9 2017.28   375.7 2013.94
   496.1 1956.66   556.5 1932.74   596.8 1914.74   614.5 1909.92     627 1908.24
     637 1909.93   639.5  1911.5   667.2 1930.22   737.7 1972.77     788 2008.92
   838.3 2040.86   908.7 2089.81   948.9 2112.45     989  2133.1  1039.2 2154.21
  1049.3  2157.1  1109.5 2160.97  1179.7 2174.21    1240 2190.25  1370.5 2230.85
#Mann= 3 , 0 , 0
       0     .08       0   614.5    .045       0   639.5     .08       0
Bank Sta=614.5,639.5
XS Rating Curve= 0 ,0
Exp/Cntr=0.3,0.1

Type RM Length L Ch R = 1 ,7336    ,481.5,472.7,463.9
XS GIS Cut Line= 4
     1848761.886      157083.731      1848486.47      157164.776
     1848048.481      157542.348     1847812.802      157790.766
#Sta/Elev= 30
     9.9 2130.54    59.4 2103.27      99 2075.17   108.9 2069.22   128.7 2060.73
   158.4 2050.54   178.2 2041.74   267.3 1994.58     307 1975.07   336.9    1962
   346.9 1960.28   356.9 1960.75   416.7 1972.43   436.6 1974.16   456.6 1973.91
   466.6 1971.19   476.5 1966.61   506.4  1949.2   586.2 1907.27   613.6 1901.47
   626.1 1900.88   638.6  1904.4   705.8 1939.09   745.7 1957.24   865.4 1990.97
   885.5 1999.38   915.7 2014.38     956 2029.09  1046.6 2054.88  1207.8 2091.77
#Mann= 3 , 0 , 0
       0     .08       0   613.6    .045       0   638.6     .08       0
Bank Sta=613.6,638.6
XS Rating Curve= 0 ,0
Exp/Cntr=0.3,0.1

Type RM Length L Ch R = 1 ,6863.3  ,416.1,420.8,425.5
XS GIS Cut Line= 4
     1848341.486      156669.701     1848053.492      156818.722
     1847780.954      157274.821     1847666.299      157606.045
#Sta/Elev= 30
     9.8 2220.32    39.3 2209.67    88.4 2197.58   108.1  2189.5   206.4 2127.26
     226 2111.45   265.3    2075     285  2058.1   304.6 2043.58   354.3 2011.39
   414.5 1976.74   544.8 1910.07   554.8 1905.23   582.4 1895.48   594.9 1893.29
   607.4 1896.17     635 1908.89   745.3 1954.36   765.4 1956.62   865.6 1956.01
   875.6 1956.85   885.6 1959.57   905.7  1969.1   945.7 1991.28  1005.8 2028.72
  1035.8 2045.89  1065.9 2060.24    1126 2085.97    1146 2095.96  1206.1 2139.05
#Mann= 3 , 0 , 0
       0     .08       0   582.4    .045       0   607.4     .08       0
Bank Sta=582.4,607.4
XS Rating Curve= 0 ,0
Exp/Cntr=0.3,0.1

Type RM Length L Ch R = 1 ,6442.5  ,500.3,476.6,452.8
XS GIS Cut Line= 4
     1848023.599      156555.098     1847806.432      156593.265
     1847477.042      156951.652     1847354.185      157319.409
#Sta/Elev= 30
      10 2161.41   220.5  2034.9   329.8 1950.13   369.5 1913.68   379.4 1906.38
   389.4 1900.66   399.3 1896.77   409.2 1894.03   466.3 1884.33   478.8 1883.25
   491.3 1883.59   528.4 1886.99   538.4 1889.07     598 1911.38   627.8 1921.81
   637.7 1924.62   647.7 1926.19   657.6 1925.75   687.4 1920.49   697.3 1919.51
   707.3 1920.18   727.1  1925.6   786.8 1945.13   816.6 1953.47   856.4 1961.97
   896.2  1968.8   935.9 1976.99   995.6 1987.98  1025.4 1995.24    1095 2015.36
#Mann= 3 , 0 , 0
       0     .08       0   466.3    .045       0   491.3     .08       0
Bank Sta=466.3,491.3
XS Rating Curve= 0 ,0
Exp/Cntr=0.3,0.1

Type RM Length L Ch R = 1 ,5965.9  ,445.7,466.3,486.8
XS GIS Cut Line= 4
     1847258.639       156077.32     1847203.707      156409.102
     1847271.379      156873.531     1847188.532      157091.231
#Sta/Elev= 30
     9.9 2148.15    59.3 2115.11   138.5 2065.74   197.8 2030.85   227.5 2014.29
   286.8 1984.47   326.4 1966.46   376.2 1946.52   426.2 1927.91   436.2 1923.38
   496.1 1891.11     516 1878.93   523.5 1876.53     536 1875.29   548.5 1876.15
   635.9 1880.73   675.8 1883.93   685.8 1885.41   695.8 1888.26   705.8 1892.71
   805.6 1950.07   854.2 1984.93   883.3 2008.99     893 2015.27   931.8 2034.08
   960.9  2050.3   970.6 2056.96  1009.4 2087.16  1019.2 2093.62  1038.6 2103.41
#Mann= 3 , 0 , 0
       0     .08       0   523.5    .045       0   548.5     .08       0
Bank Sta=523.5,548.5
XS Rating Curve= 0 ,0
Exp/Cntr=0.3,0.1

Type RM Length L Ch R = 1 ,5499.7  ,414.5,419,423.5
XS GIS Cut Line= 4
     1847143.985       156077.32     1846949.768      156302.035
     1846659.889      156765.246     1846589.822      157013.664
#Sta/Elev= 30
     9.9  2111.2    79.2 2059.01   148.5 2008.35   178.2 1984.09   188.1 1976.84
   207.9 1964.71   237.6  1949.3   287.1 1929.91   356.6  1908.1   386.4 1899.44
   416.2 1891.67     456 1882.41   475.8 1878.47   525.5 1870.29   542.8 1866.13
   555.3 1864.36   567.8 1865.61   595.1 1873.62   614.9 1880.99   644.7 1894.28
   704.4 1919.47     754 1942.53   773.9  1950.2   783.8 1954.75   843.5 1991.05
   893.1 2017.83   942.7 2041.59  1022.1 2086.64    1042 2095.68  1101.6 2116.08
#Mann= 3 , 0 , 0
       0     .08       0   542.8    .045       0   567.8     .08       0
Bank Sta=542.8,567.8
XS Rating Curve= 0 ,0
Exp/Cntr=0.3,0.1

Type RM Length L Ch R = 1 ,5080.7  ,483.6,456.1,428.5
XS GIS Cut Line= 4
     1846946.525      155898.969     1846746.017       155965.86
     1846322.295      156446.762      1846220.38      156752.507
#Sta/Elev= 30
    10.1 2079.12    50.3 2054.48   110.7 2021.94   140.9 2008.06   211.4 1981.51
   251.4 1963.49   301.5 1948.02   491.8 1873.49   521.8 1866.06   569.4  1858.3
   581.9 1857.78   594.4 1859.79     622  1867.7     632 1871.78     642 1877.45
     652 1884.72     662 1893.87   692.1 1925.11   702.1 1933.93   712.1 1941.34
   772.2 1977.48   862.4 2035.84   872.5 2041.94   882.5 2046.54   902.7 2053.98
   932.9 2061.09   983.2 2068.23    1084 2089.26  1114.2 2096.64  1174.6 2114.52
#Mann= 3 , 0 , 0
       0     .08       0   569.4    .045       0   594.4     .08       0
Bank Sta=569.4,594.4
XS Rating Curve= 0 ,0
Exp/Cntr=0.3,0.1

Type RM Length L Ch R = 1 ,4624.6  ,417.4,420.2,422.9
XS GIS Cut Line= 4
     1846067.508      155516.788     1846088.728      155791.976
      1846233.12       156287.52     1846130.604      156555.856
#Sta/Elev= 30
     9.9 2128.21    29.6 2114.99      69 2095.26   177.4 2036.91   226.7 2011.64
   246.4  1999.6   295.9 1966.21   345.5 1934.28     415 1893.38   464.6 1866.71
   484.5 1858.56   501.7 1853.19   514.2 1851.87   526.7    1853   603.6 1864.89
     673 1868.68     683 1870.28   692.9 1874.18   702.8 1879.78   792.2 1937.57
     812 1948.11   821.9 1952.44   831.8 1955.29   861.5 1960.52   920.9 1966.59
   960.5 1974.84    1020 1980.24  1039.8 1982.73  1069.5 1988.52  1079.4  1991.8
#Mann= 3 , 0 , 0
       0     .08       0   501.7    .045       0   526.7     .08       0
Bank Sta=501.7,526.7
XS Rating Curve= 0 ,0
Exp/Cntr=0.3,0.1

Type RM Length L Ch R = 1 ,4204.5  ,446.3,464.1,482
XS GIS Cut Line= 4
     1845774.502      155644.181     1845736.284      155975.405
     1845814.113      156384.013     1845806.351       156688.81
#Sta/Elev= 30
    10.1 2103.42    40.4 2087.63    90.9 2065.57   111.1 2054.32   131.3 2040.02
   161.7 2016.93   202.1 1989.09   242.5 1963.37   282.9 1935.63   333.4 1904.88
   353.2 1895.59   392.8 1880.46     482 1849.83   491.9 1847.15     519 1844.95
   531.5 1844.69     544 1846.02   551.3 1847.58   610.7 1865.28   719.7 1905.13
   739.5  1913.8   778.9 1935.91   818.2 1959.41   828.1 1965.63   857.6 1986.76
   877.2 1999.03   916.6 2017.55   985.4 2052.93  1034.6  2086.4  1054.3 2100.56
#Mann= 3 , 0 , 0
       0     .08       0     519    .045       0     544     .08       0
Bank Sta=519,544
XS Rating Curve= 0 ,0
Exp/Cntr=0.3,0.1

Type RM Length L Ch R = 1 ,3740.3  ,166.8,172.2,177
XS GIS Cut Line= 4
     1845569.866      155684.377     1845468.883      155850.587
     1845252.188      156293.889     1845040.187      156431.404
#Sta/Elev= 30
     9.7 2060.98    48.6 2037.44     107 1989.85   184.8 1934.79   214.6 1915.84
   244.8 1899.25     275 1884.49   345.5 1853.77     406 1836.27     416 1834.72
   453.9 1833.06   466.4 1832.36   478.9 1833.66   486.5 1836.44   506.7 1848.32
   546.9 1867.72   577.1 1883.85   607.4 1901.73   637.6  1921.8   657.7 1937.05
   677.8 1955.09   728.3 2009.34   748.6 2028.44   768.8 2044.45     789  2056.8
   819.3 2069.75   859.7 2080.79     880 2083.46   900.2 2083.86   940.6 2080.48
#Mann= 3 , 0 , 0
       0     .08       0   453.9    .045       0   478.9     .08       0
Bank Sta=453.9,478.9
XS Rating Curve= 0 ,0
Exp/Cntr=0.3,0.1

Type RM Length L Ch R = 1 ,3568.2  ,256.6,234.6,212.8
XS GIS Cut Line= 4
     1845455.188      155518.687     1845320.696      155851.181
     1845152.581      156075.334     1845021.825      156306.959
#Sta/Elev= 30
      10 2075.86    49.8 2067.19    99.6 2052.67   139.5 2038.87   169.4 2026.53
   179.3  2021.6   189.3 2015.63   199.3 2008.02   209.2 1998.54   229.1 1976.75
   239.1 1966.52     259 1950.51   288.9    1930   328.8 1903.96   338.7 1898.47
   358.7 1889.95   418.7 1869.93   438.7 1862.14   488.8 1840.55   516.3 1831.25
   528.8 1828.86   541.3 1829.46   578.8 1839.79   658.6 1865.39   668.4 1870.35
   678.3 1876.39   737.4 1917.01   766.9 1935.34   885.1 2002.54   904.8 2012.07
#Mann= 3 , 0 , 0
       0     .08       0   516.3    .045       0   541.3     .08       0
Bank Sta=516.3,541.3
XS Rating Curve= 0 ,0
Exp/Cntr=0.3,0.1

Type RM Length L Ch R = 1 ,3333.6  ,494.5,518.1,539.5
XS GIS Cut Line= 4
     1845234.462      155454.827     1845003.145      155716.689
     1845055.448      156094.013     1844856.635      156336.322
#Sta/Elev= 30
      10 2079.88    59.9 2067.21   109.8 2050.37   149.7 2033.17   209.6 2001.58
   229.6 1989.32   249.6 1974.15   259.6 1965.62   299.5  1927.8   319.4 1910.04
   329.4 1902.08   349.4 1890.39   379.5 1877.87   409.5 1867.41   439.6 1857.93
   479.7 1847.35   499.8 1841.08   537.4 1825.02   549.9 1823.15   562.4 1824.57
     600 1831.26   700.3 1861.15   710.3 1864.93   740.4 1881.33   801.1 1909.99
   841.5 1926.91   892.1 1946.68   912.3    1957   942.7 1975.65  1043.8 2041.69
#Mann= 3 , 0 , 0
       0     .08       0   537.4    .045       0   562.4     .08       0
Bank Sta=537.4,562.4
XS Rating Curve= 0 ,0
Exp/Cntr=0.3,0.1

Type RM Length L Ch R = 1 ,2815.5  ,195,219.5,244.2
XS GIS Cut Line= 4
     1845145.061      155398.998     1844787.201      155497.678
     1844436.868      155930.817     1844460.364       156148.43
#Sta/Elev= 30
      10 2076.17    30.1 2065.56    90.3 2037.57   170.6 2005.41   250.8 1967.91
   331.1 1939.04   371.2 1927.55     421 1925.86   470.7 1922.44   480.6 1921.57
   490.6 1918.39   500.5 1914.05   530.4 1897.96     610 1853.23   659.7 1824.42
   679.6 1810.07     687 1806.32   689.5 1805.05   699.5 1803.93     712 1804.81
   749.2 1814.35   848.7 1846.57   858.7 1847.41   888.5 1846.09   928.3 1846.39
   968.1 1848.33     978 1850.21  1087.5  1896.1  1117.3 1909.92  1147.2 1925.71
#Mann= 3 , 0 , 0
       0     .08       0     687    .045       0     712     .08       0
Bank Sta=687,712
XS Rating Curve= 0 ,0
Exp/Cntr=0.3,0.1

Type RM Length L Ch R = 1 ,2596    ,288.6,297.5,306.3
XS GIS Cut Line= 4
     1845152.581      155361.779     1844566.047      155574.725
     1844334.422      155574.725     1844143.892      155858.652
#Sta/Elev= 30
    10.1 2066.16    30.2 2057.97    50.3 2048.47   100.6 2027.68   191.2 1997.75
   261.7 1967.04   281.8  1959.1   362.3  1933.5   422.7 1918.47   493.2 1897.26
   503.2 1893.63   543.5  1876.7   674.3 1817.61   704.6 1803.33   712.2 1800.48
   714.6 1799.58   724.7 1798.44   737.2 1799.91     765 1806.24   855.6 1821.97
     916 1836.53   946.1 1841.95   976.3 1844.41  1086.9 1845.62    1107 1846.82
  1127.2 1852.04  1147.3 1858.94  1167.4 1868.28  1187.5 1878.49  1197.5 1882.55
#Mann= 3 , 0 , 0
       0     .08       0   712.2    .045       0   737.2     .08       0
Bank Sta=712.2,737.2
XS Rating Curve= 0 ,0
Exp/Cntr=0.3,0.1

Type RM Length L Ch R = 1 ,2298.5  ,394.9,397,399.1
XS GIS Cut Line= 4
     1845127.715      155305.182     1844816.351      155399.138
     1844424.083      155268.382     1844191.646      155143.048
#Sta/Elev= 30
     9.9 2027.46    39.4 2015.91    78.8 2001.82   108.4 1992.23   167.5 1974.22
   216.8 1958.12   236.5 1950.42   285.8 1929.22   325.2 1913.79     416 1864.45
   516.8 1808.39   534.6 1797.86     537 1796.51   547.1 1793.64   559.6  1794.4
   577.4 1797.95   587.4 1798.93   607.6 1799.23     648  1798.8   668.1 1800.32
   688.3 1804.14   698.4 1807.16   708.5 1810.94   728.6 1820.79   758.3 1837.74
   787.6 1852.73   797.4 1858.42   836.5 1883.63   953.9 1960.75  1002.8 1995.48
#Mann= 3 , 0 , 0
       0     .08       0   534.6    .045       0   559.6     .08       0
Bank Sta=534.6,559.6
XS Rating Curve= 0 ,0
Exp/Cntr=0.3,0.1
